--- 2953_ras.prj (project) ---

Proj Title=2953
Current Plan=p01
Default Exp/Contr=0.3,0.1
English Units
Geom File=g01
Flow File=f01
Plan File=p01
Y Axis Title=Elevation
X Axis Title(PF)=Main Channel Distance
X Axis Title(XS)=Station
BEGIN DESCRIPTION:
RFD model 2953 exported to HEC-RAS
END DESCRIPTION:

--- 2953_ras.p01 (plan) ---

Plan Title=Plan 01
Program Version=4.10
Short Identifier=Plan 01
Geom File=g01
Flow File=f01
Subcritical Flow
Calc Critical at every XS
Secant Critical Depth

--- 2953_ras.f01 (steady flow) ---

Flow Title=Flow 01
Program Version=5.01
Number of Profiles= 6
Profile Names=10yr,25yr,50yr,100yr,100plus,500yr
River Rch & RM=2953,118,95981.72
 2632.23 3992.42 5217.25 6236.08 9104.6810086.76
River Rch & RM=2953,118,95734.86
 2656.49  4030.8  5268.8 6299.13 9196.7310179.36
River Rch & RM=2953,118,95487.99
 2661.43 4038.68 5279.41 6312.17 9215.7610198.66
River Rch & RM=2953,118,95241.13
 2668.75 4050.31 5295.09  6331.4 9243.8410227.06
River Rch & RM=2953,118,94994.27
    2696  4093.6 5353.37 6402.84 9348.15 10332.3
River Rch & RM=2953,118, 94747.4
 2699.36 4098.95  5360.6 6411.71  9361.110345.43
River Rch & RM=2953,118,94500.54
    2726 4141.27 5417.59 6481.58 9463.1110448.18
River Rch & RM=2953,118,94253.67
 2732.44 4151.54 5431.44  6498.6 9487.9610473.31
River Rch & RM=2953,118,94006.81
 2740.41 4164.25  5448.6 6519.68 9518.7410504.43
River Rch & RM=2953,118,93759.94
 2750.11 4179.75 5469.55 6545.45 9556.3510542.53
River Rch & RM=2953,118,93513.08
 2751.65 4182.21 5472.87 6549.52 9562.3110548.54
River Rch & RM=2953,118,93266.22
 2755.94 4189.09 5482.18    6561 9579.0510565.56
River Rch & RM=2953,118,93019.35
 2761.23 4197.57 5493.68 6575.16 9599.7310586.58
River Rch & RM=2953,118,92772.74
 2764.74  4203.2 5501.31 6584.57 9613.4710600.58
River Rch & RM=2953,118,92526.13
 2768.02 4208.46 5508.43 6593.34 9626.2710613.57
River Rch & RM=2953,118,92279.52
 2782.32  4231.3 5539.27 6631.25 9681.6210669.47
River Rch & RM=2953,118,92032.91
 2783.32  4232.9 5541.44 6633.93 9685.5310673.46
River Rch & RM=2953,118, 91786.3
 9020.5913781.6818115.0421726.2831720.3729644.06
River Rch & RM=2953,118,91218.95
 9034.6713804.4718146.1421764.7831776.5829692.78
River Rch & RM=2953,118,90892.46
 9512.2714570.2419184.63 23043.633643.6531283.99
River Rch & RM=2953,118,90459.09
 9515.2814575.1419191.31 23051.933655.7731294.45
River Rch & RM=2953,118, 89874.6
 9537.6114611.55 19241.223113.8733746.2431372.83
River Rch & RM=2953,118,89168.43
 9713.4414894.4319625.6623588.2134438.7931962.16
River Rch & RM=2953,118,88370.11
 9556.1314641.6919282.4523165.07   3382131437.44
River Rch & RM=2953,118,87882.09
 9563.3314653.3619298.3923184.8133849.8331462.22
River Rch & RM=2953,118,87394.06
 9574.3714671.2419322.7723214.9933893.8831500.04
River Rch & RM=2953,118,86906.03
 9607.6814725.0619396.1123305.6834026.2931613.38
River Rch & RM=2953,118,86418.01
 9711.7514891.6919621.9223583.5734432.0131956.32
River Rch & RM=2953,118,85929.98
 9743.0714942.1919690.6423668.4634555.95 32061.9
River Rch & RM=2953,118,85441.95
 9756.3114963.6419719.9123704.6934608.85 32107.2
River Rch & RM=2953,118,84953.93
 9790.0215018.3919794.7523797.4934744.3332223.57
River Rch & RM=2953,118, 84465.9
  9799.215033.2919815.1223822.7534781.2132255.22
River Rch & RM=2953,118,83893.21
 9811.1915052.7619841.7323855.7334829.3632296.54
River Rch & RM=2953,118,83489.85
 9990.6215344.1620240.04 24349.635550.4232914.52
River Rch & RM=2953,118,83001.82
  9995.115351.4320249.9724361.9135568.3932929.89
River Rch & RM=2953,118, 82529.1
10005.5815368.4320273.1924390.6835610.3932965.76
River Rch & RM=2953,118,82025.77
10066.3215466.3820406.5424555.4435850.9533169.76
River Rch & RM=2953,118,81537.74
10072.6915476.7120420.6324572.8935876.4333191.48
River Rch & RM=2953,118,81049.72
10085.2315497.1220448.5724607.5835927.0733234.89
River Rch & RM=2953,118,80561.69
10114.7715545.2720514.5424689.5436046.7333337.58
River Rch & RM=2953,118,80073.66
10127.89 15566.720543.9324726.0936100.0933383.46
River Rch & RM=2953,118,79585.64
10138.9515584.7920568.77   2475736145.2233422.32
River Rch & RM=2953,118,79183.71
10152.0115606.1520598.0824793.4736198.4733468.16
River Rch & RM=2953,118,78781.77
10155.6215612.06 20606.224803.5836213.2333480.89
River Rch & RM=2953,118,78379.84
10163.8715625.5820624.8124826.78 36247.133510.16
River Rch & RM=2953,118,77977.91
10180.4815652.7820662.1624873.29   3631533568.67
River Rch & RM=2953,118,77133.19
10230.9815735.3720775.5325014.3836520.9933745.86
River Rch & RM=2953,118,76690.39
10241.6715752.9320799.7125044.5436565.0233783.92
River Rch & RM=2953,118, 76247.6
10255.7115776.0220831.49 25084.236622.93   33834
River Rch & RM=2953,118, 75804.8
10963.7316902.47 22352.526950.0239347.0336084.07
River Rch & RM=2953,118, 75193.4
10971.4616915.1622369.97 26971.839378.8336111.26
River Rch & RM=2953,118, 74013.4
11106.7117137.0122675.1227352.2239934.2536585.11
River Rch & RM=2953,118,73139.32
 11198.417287.1722881.4827609.2940309.5736904.16
River Rch & RM=2953,118,72702.28
11200.8217291.1522886.9727616.1540319.5836912.74
River Rch & RM=2953,118,72265.24
11237.3717351.4722970.2627720.3240471.6637043.11
River Rch & RM=2953,118,71644.44
11260.3717389.4323022.6527785.8340567.3137125.03
River Rch & RM=2953,118,69990.13
11339.81 17520.923204.4828013.5440899.7737410.59
River Rch & RM=2953,118,69540.05
11799.7318269.2424229.1129285.89 42757.438968.61
River Rch & RM=2953,118,69089.97
11806.12 18279.824243.7229304.1942784.1238991.39
River Rch & RM=2953,118,68639.89
11822.5718307.0224281.3629351.3442852.9639050.11
River Rch & RM=2953,118,68189.81
11828.6218317.0424295.2129368.6842878.2739071.68
River Rch & RM=2953,118,67739.73
11837.7818332.2224316.2329395.0542916.7739104.61
River Rch & RM=2953,118,67289.65
11860.4318369.9624368.63 29460.943012.9139187.21
River Rch & RM=2953,118,66839.57
11881.3118404.6324416.69 29521.243100.9539262.56
River Rch & RM=2953,118,66360.96
11899.16 18434.324457.8229572.8343176.33 39327.1
River Rch & RM=2953,118,65882.36
11908.9418450.62 24480.529601.3643217.9939362.94
River Rch & RM=2953,118,65403.75
11916.4518463.13 24497.929623.2543249.9439390.41
River Rch & RM=2953,118,64925.15
12188.0518908.4825110.5930387.2244365.3440328.77
River Rch & RM=2953,118,64446.54
12466.7419371.58 25752.831193.5245542.5441331.29
River Rch & RM=2953,118,63967.94
12477.0919388.9925777.1331224.2445587.3941369.95
River Rch & RM=2953,118,63489.33
12491.1619412.6825810.2331266.0845648.4741422.64
River Rch & RM=2953,118,63010.73
12503.3519433.3825839.2931302.94 45702.341469.47
River Rch & RM=2953,118,62532.12
12576.5519555.7126009.5431517.3346015.31 41737.1
River Rch & RM=2953,118,62053.52
12581.2419563.95 26021.331532.4846037.4241756.94
River Rch & RM=2953,118,61574.92
12613.1519619.0426099.3831632.3246183.1941885.82
River Rch & RM=2953,118,61188.63
12618.6119628.6326113.1331650.0546209.0741909.13
River Rch & RM=2953,118,60617.71
12646.0119675.5326179.29 31734.346332.0842016.88
River Rch & RM=2953,118,59835.38
12658.3419697.0326209.9131773.63 46389.542068.09
River Rch & RM=2953,118,59137.85
 12701.319771.0126314.63 31907.446584.8142240.16
River Rch & RM=2953,118,57887.94
12879.5920075.0526742.7132451.8147379.6442932.68
River Rch & RM=2953,118, 56935.3
 12894.520102.1726782.2632503.5547455.1943002.49
River Rch & RM=2953,118,56178.13
12900.1520112.6426797.6532523.8147484.7743030.18
River Rch & RM=2953,118,55384.16
12906.8420125.0326815.8832547.8247519.8243063.04
River Rch & RM=2953,118,55042.37
12908.01 20127.226819.0832552.0447525.98 43068.8
River Rch & RM=2953,118,54243.43
13355.8120928.3727977.4234057.5949724.0945066.68
River Rch & RM=2953,118,53296.16
13372.1620958.9328022.62 34117.449811.4145148.76
River Rch & RM=2953,118, 52348.9
13528.7721243.73 28438.134661.4250605.6745878.71
River Rch & RM=2953,118,51744.59
13550.2921284.4328498.6534741.9350723.22   45990
River Rch & RM=2953,118,50622.25
13590.2621360.3828611.9434892.8750943.5946199.36
River Rch & RM=2953,118,50065.56
13596.2521371.8428629.11 34915.850977.0746231.32
River Rch & RM=2953,118,48693.52
13678.1921529.3728865.4435232.0451438.77 46673.4
River Rch & RM=2953,118,46665.31
13695.9421563.29 28916.235299.8351537.7546767.76
River Rch & RM=2953,118,45718.05
13712.3621594.4828962.7335361.8451628.2946853.68
River Rch & RM=2953,118,44770.78
13720.2921609.58 28985.335391.9551672.25 46895.5
River Rch & RM=2953,118,43823.52
13902.0221949.3229488.32 36058.552645.4147807.47
River Rch & RM=2953,118,42876.25
13925.9821995.1729556.9936150.3352779.4847935.21
River Rch & RM=2953,118,41805.52
 13934.922012.2329582.54 36184.552829.3847982.74
River Rch & RM=2953,118,40473.47
13951.2722043.5529629.4736247.2552920.9948070.01
River Rch & RM=2953,118,39561.03
13963.7522067.5529665.5136295.5252991.4548137.35
River Rch & RM=2953,118,38570.99
14008.7822154.1329795.5436469.7453245.8248380.46
River Rch & RM=2953,118,37211.91
14021.0222177.7529831.0636517.3953315.3948447.08
River Rch & RM=2953,118,35908.86
14040.2722214.9229887.0136592.4953425.0448552.17
River Rch & RM=2953,118,33893.97
14127.8922383.8830141.1436933.4553922.8449028.62
River Rch & RM=2953,118,32741.88
14280.0122677.6430583.5137527.5554790.2349859.15
River Rch & RM=2953,118,32562.05
14284.1222685.5730595.4237543.5454813.5749881.46
River Rch & RM=2953,118,31149.73
14294.9722706.4530626.8337585.68 54875.149940.22
River Rch & RM=2953,118,28747.58
14316.3322747.3530688.1937667.8754995.0950054.39
River Rch & RM=2953,118,25833.52
 14401.622909.9730931.6837993.5455470.5750505.18
River Rch & RM=2953,118,23179.28
14483.5823066.4231166.0438307.1655928.4550939.28
River Rch & RM=2953,118,19705.56
14509.39 23115.231238.7838404.1656070.0751072.52
River Rch & RM=2953,118,17884.19
14826.7523715.2532133.9939598.6757814.0652712.01
River Rch & RM=2953,118, 13275.9
14848.8823757.3432196.9839682.9357937.0952828.04
River Rch & RM=2953,118,8529.917
14898.5223852.6332340.2939875.3658218.0353094.86
River Rch & RM=2953,118,5187.372
14898.81 23853.232341.1439876.51 58219.753096.45
Boundary for River Rch & Prof#=2953,118,1
Up Type= 0
Dn Type= 2
Boundary for River Rch & Prof#=2953,118,2
Up Type= 0
Dn Type= 2
Boundary for River Rch & Prof#=2953,118,2
Up Type= 0
Dn Type= 2
Boundary for River Rch & Prof#=2953,118,2
Up Type= 0
Dn Type= 2
Boundary for River Rch & Prof#=2953,118,2
Up Type= 0
Dn Type= 2
Boundary for River Rch & Prof#=2953,118,2
Up Type= 0
Dn Type= 2

--- 2953_ras.g01 (geometry) ---

Geom Title=2953
Program Version=4.10

River Reach=2953,118
Reach XY= 30
  450583.8821069781680.282259256447366.312662363784429.448925942
 446742.28488487783408.337814823447688.726062417782713.752898097
444832.137865424782666.209559739445349.269838333 781650.60633336
443786.769838303781003.523000047441629.680599898781732.711119264
441074.408727169779581.578555509434320.311505139779990.398000017
432284.845472455777957.863022745430981.422616065778142.898000062
429657.255949408776260.398000017430432.327875316774902.268053621
429030.867060512773796.925777748430190.450394005770445.502167016
429474.660187244769488.201440886429261.630949408771054.877166644
427969.130949885770979.738277793427943.575394064768735.293833435
426930.389627218768873.618191093426750.924930871  765958.5692963
 428010.92493096762939.958185196425263.702708662761340.513740718
  423321.5499309762344.263740733422211.133264661761068.013740763
420127.799931169760940.097074091412807.084616393765365.125400633
410595.950357169765479.407808051409320.394801617767677.741141915

Type RM Length L Ch R = 1 ,95981.72,246.864100,246.864100,246.864100
XS GIS Cut Line= 6
450570.813024417781479.700435348 450578.89767594781592.688833196
450583.933315084781702.086296391450587.375717298781740.466112693
450598.374036704781807.399623867450616.419353421781877.917790038
#Sta/Elev= 30
9799.005753.93519804.318752.01949814.344750.47219834.395 749.7829854.446750.0059
9894.548747.67929904.574744.80089914.596741.12569924.606738.54119954.637726.0702
9974.658723.49449984.669721.578110004.69722.8734 10014.7725.371510024.72734.7141
10034.76740.2344 10044.8740.904110054.84746.575410064.92760.558810075.06770.9122
10085.19 780.00410095.33781.903510105.46780.917210115.59780.974710125.73  784.37
10136.01 792.51810146.33 798.91510156.65802.585810177.29811.146810200.95818.5996
#Mann= 3 , 0 , 0
9799.005    0.12       09799.005    0.12       010200.95    0.12       0
#XS Ineff= 2 , 0
       0                               0
Bank Sta=9799.005,10200.95
Exp/Cntr=0.3,0.1

Type RM Length L Ch R = 1 ,95734.86,246.864100,246.864100,246.864100
XS GIS Cut Line= 6
450280.985220192781526.371843014450297.729977736781609.583990199
450315.397704607781662.583609721450346.974537055781727.099615692
450400.960777411781814.798312559450438.674763751781892.394632539
#Sta/Elev= 30
9799.053829.19739807.855828.35289818.055825.54139828.255821.28989858.857804.0126
9869.057 797.5429879.258790.59069909.723 767.5139921.057757.84669942.524741.9612
9953.639731.6548 9975.87719.77469986.986709.86969998.101708.118610007.36707.9008
10011.67708.399710021.08712.202810026.44716.262610056.82 735.02710068.73736.4355
10080.38745.842510091.89752.458210103.41761.109610114.92763.980810126.03763.3461
10137.15765.096210148.27770.725810159.39774.326910181.63776.729310200.97780.5707
#Mann= 3 , 0 , 0
9799.053    0.12       09799.053    0.12       010200.97    0.12       0
#XS Ineff= 2 , 0
       0                               0
Bank Sta=9799.053,10200.97
Exp/Cntr=0.3,0.1

Type RM Length L Ch R = 1 ,95487.99,246.864100,246.864100,246.864100
XS GIS Cut Line= 6
450183.749319639781563.984145836 450182.64822742781697.981266624
 450167.44673815781732.185470252450125.434450164 781783.38427067
450109.524018131781830.594721875450117.993128176781942.519844777
#Sta/Elev= 30
9799.109807.49819810.173797.91189820.217790.45349830.261 781.5319839.875775.4272
9850.312768.1117 9860.32758.79089870.328751.08979890.345740.76669900.354734.1795
9910.452728.48959941.248717.56979951.878714.68979955.776712.56869974.898697.3996
9987.581696.242310005.31696.801310020.51700.935210027.73701.970110039.56702.8444
10061.34 706.04510071.67708.5445 10092.2712.556110102.25  714.0110142.34723.3357
 10162.5729.838610172.63730.720910187.37733.968910193.14735.528210200.85738.3263
#Mann= 3 , 0 , 0
9799.109    0.12       09799.109    0.12       010200.85    0.12       0
#XS Ineff= 2 , 0
       0                               0
Bank Sta=9799.109,10200.85
Exp/Cntr=0.3,0.1

Type RM Length L Ch R = 1 ,95241.13,246.864200,246.864200,246.864200
XS GIS Cut Line= 6
449821.978451055781668.431789129449861.439081494781727.293348995
449904.664085032781785.994629699449965.830168137781858.457839036
450001.640773696781904.713799992450060.485599129781991.401951241
#Sta/Elev= 30
9799.022772.81959822.407762.85979831.009760.77749840.365756.69579855.087750.1347
9875.893739.27239891.876734.60589909.623728.50449916.714724.54299929.132714.8339
9943.331704.39289954.222695.69829959.557692.1445 9966.92689.24479975.782687.1501
9991.547686.759810006.39688.482910019.73694.797410045.96703.605510052.66706.6511
10071.25716.5971 10083.9720.963810102.16724.4501 10120.7 726.47710144.87731.9617
10156.96732.543810169.04736.189610181.13738.709710193.22739.835410200.95742.3841
#Mann= 3 , 0 , 0
9799.022    0.12       09799.022    0.12       010200.95    0.12       0
#XS Ineff= 2 , 0
       0                               0
Bank Sta=9799.022,10200.95
Exp/Cntr=0.3,0.1

Type RM Length L Ch R = 1 ,94994.27,246.864100,246.864100,246.864100
XS GIS Cut Line= 6
449619.133856632781896.004736269449678.157907447781944.715961242
449730.664433589781981.672954212449761.860076783 782000.31652111
449853.653260202   782048.821209449955.608230891782113.977366104
#Sta/Elev= 30
9799.047738.35689806.652734.82799832.584725.36449845.549718.87959860.311714.9547
9876.069713.78979883.942712.09839896.171708.20989910.816705.96299944.835695.4881
9956.484690.62959968.134684.62659976.126683.62669990.891679.823610013.29679.5806
10024.48684.568810035.69697.611510051.63712.360110070.06726.305310081.55733.0375
10091.79742.638310116.74769.739410128.46780.382110140.19789.324810148.72791.6609
10166.76791.030410176.22794.0212 10184.8800.980110200.26819.095310200.99819.3382
#Mann= 3 , 0 , 0
9799.047    0.12       09799.047    0.12       010200.99    0.12       0
#XS Ineff= 2 , 0
       0                               0
Bank Sta=9799.047,10200.99
Exp/Cntr=0.3,0.1

Type RM Length L Ch R = 1 , 94747.4,246.864100,246.864100,246.864100
XS GIS Cut Line= 6
449489.027472657782120.447950493449549.716383445782160.609453042
449634.789389116782206.648332408449686.861402011782236.690163751
449727.044333761782254.866542336449846.108119034782302.401998983
#Sta/Elev= 30
9799.049748.21339807.297741.69379818.202734.47379825.418730.80499842.185725.3284
9854.176 723.4789877.831 712.9599911.942700.39769934.683690.2037 9944.08686.7866
9968.799682.23939980.388674.37929991.978669.901510003.56669.102310015.05 669.407
10026.54674.507110037.61683.083610070.53  710.7110081.34715.603410092.11717.1194
10100.11721.203510102.88 723.29210113.65735.143510124.41744.119410145.95758.8453
10156.72767.371710167.48774.052210189.02775.706610199.79777.179610200.98777.8998
#Mann= 3 , 0 , 0
9799.049    0.12       09799.049    0.12       010200.98    0.12       0
#XS Ineff= 2 , 0
       0                               0
Bank Sta=9799.049,10200.98
Exp/Cntr=0.3,0.1

Type RM Length L Ch R = 1 ,94500.54,246.864100,246.864100,246.864100
XS GIS Cut Line= 6
449419.014530171782363.859035795449464.714731319782402.737140583
449517.945056636782432.206094068449565.958829385782450.192426988
 449697.51190845782490.274015841449783.836411534782522.457044157
#Sta/Elev= 30
9799.065711.59369829.766698.29649846.432693.05839859.138690.38359871.177688.8135
9894.554684.10379905.665682.49619927.583675.40739938.261673.0527 9948.94671.5085
9959.618671.34599970.297669.45599980.767664.52849991.214661.485610001.65661.7328
10012.11663.034810022.57669.501810043.48690.235110053.94698.720410064.39699.5709
10074.85702.107510085.31714.069910095.76724.652810106.22728.892910116.84732.4367
10148.85740.404910159.53740.8907 10170.2738.649110180.87735.433610200.97730.6668
#Mann= 3 , 0 , 0
9799.065    0.12       09799.065    0.12       010200.97    0.12       0
#XS Ineff= 2 , 0
       0                               0
Bank Sta=9799.065,10200.97
Exp/Cntr=0.3,0.1

Type RM Length L Ch R = 1 ,94253.67,246.864100,246.864100,246.864100
XS GIS Cut Line= 6
449395.994109787782481.113405096449434.560388081782587.446117828
449481.651728878782685.881486542449504.547383109782724.238520482
449530.459911902782762.420727506 449586.17295693782831.582087389
#Sta/Elev= 30
9799.066677.32259824.476671.58339835.113 670.3879867.025669.33729877.663670.4523
9884.137669.72749898.938666.30459909.575665.85689920.562658.77739931.662 656.892
9953.863662.90299964.963662.20459982.303662.36479987.164661.77349998.264658.8258
10005.74658.413110009.27659.091910020.33673.464910027.84678.441110031.92680.3172
10047.35680.904610055.21683.626110066.89695.860110078.98696.5303 10102.4695.7505
10115.37695.865410127.96697.332510152.49697.295910183.77698.690810200.96700.4102
#Mann= 3 , 0 , 0
9799.066    0.12       09799.066    0.12       010200.96    0.12       0
#XS Ineff= 2 , 0
       0                               0
Bank Sta=9799.066,10200.96
Exp/Cntr=0.3,0.1

Type RM Length L Ch R = 1 ,94006.81,246.864100,246.864100,246.864100
XS GIS Cut Line= 6
449312.192327975782434.079147313449307.973764126782495.055623055
449292.707046859782545.289652277449203.409631241782704.791030992
449199.589620628782748.795497153449214.506634925782806.734061684
#Sta/Elev= 30
9799.111689.54639810.033685.28479820.033681.84939830.034678.92369840.111676.1491
9850.199673.99999860.287671.12969870.577669.10179880.869667.79649901.991664.0057
9923.843660.8289  9957.6657.56049969.604656.0287  9981.7648.72059988.434646.7311
9993.796645.865310018.36 647.00710021.79 647.89310030.25650.723110041.99656.1868
10050.02660.456110053.54661.960910064.67664.588210075.64664.813810091.52664.5555
10106.88663.571110140.83663.560910147.12663.751110188.45  666.1910200.86666.1422
#Mann= 3 , 0 , 0
9799.111    0.12       09799.111    0.12       010200.86    0.12       0
#XS Ineff= 2 , 0
       0                               0
Bank Sta=9799.111,10200.86
Exp/Cntr=0.3,0.1

Type RM Length L Ch R = 1 ,93759.94,246.864200,246.864200,246.864200
XS GIS Cut Line= 6
448892.300296112  782487.2582517448932.532086606782530.438868119
448975.120153936782569.425536537449100.857720166782663.088242535
449127.806171161782697.566762661 449170.02259435782770.605797646
#Sta/Elev= 30
9799.045742.82079803.005741.02599809.626737.08079823.294732.58659832.344732.5742
9850.629733.67769861.409733.32779864.818731.95859874.966725.09919888.524714.4201
9902.081705.39029928.315689.41959940.981679.95149953.647666.19549966.207651.8293
9974.632643.73779978.319641.05739990.432636.691110002.51636.564910010.17637.1529
10014.61637.861210027.96642.770810038.79645.3113   10065646.853310075.28648.0507
10088.45650.186110101.25 651.52510159.81654.8682 10190.9658.063610200.93659.7976
#Mann= 3 , 0 , 0
9799.045    0.12       09799.045    0.12       010200.93    0.12       0
#XS Ineff= 2 , 0
       0                               0
Bank Sta=9799.045,10200.93
Exp/Cntr=0.3,0.1

Type RM Length L Ch R = 1 ,93513.08,246.864100,246.864100,246.864100
XS GIS Cut Line= 6
448778.789272347782817.744981108448822.831924767782831.315909136
448879.945036954782843.100797368449091.681728557782866.955412727
449128.714935149782876.529137307449171.161878162782894.392424398
#Sta/Elev= 30
9799.057701.41719816.019697.80489826.483696.70819836.947697.33449857.567696.6001
9877.988695.50439888.199694.2271 9898.41686.4068 9908.55677.07099918.622 668.941
9938.766657.82769968.981642.62699979.053634.17269989.124630.42899999.197630.1906
 10009.3630.421510019.37 632.351 10029.4636.420610039.43638.203710049.47639.3422
 10059.5639.195510069.53640.101710079.56641.764510099.73646.814710130.37651.0433
10154.86653.001810161.68652.5533 10176.7648.972610183.38648.285910200.91650.1832
#Mann= 3 , 0 , 0
9799.057  0.0595       09799.057  0.0595       010200.91  0.0595       0
#XS Ineff= 2 , 0
       0                               0
Bank Sta=9799.057,10200.91
Exp/Cntr=0.3,0.1

Type RM Length L Ch R = 1 ,93266.22,246.864100,246.864100,246.864100
XS GIS Cut Line= 6
448774.594129617783006.990064148448885.892778179783054.473223569
448912.449869664783068.284594736 448950.85415334783091.577701958
449012.439752751783125.853206746449136.191447334783181.277325658
#Sta/Elev= 30
9799.032677.12979810.345671.87499832.089664.65429842.961659.66069853.833651.4712
9864.705647.54789886.449650.68749919.065647.82949930.301644.99959941.573641.1613
9952.952635.23399962.919630.93969982.202624.78359988.039623.46029999.601622.6997
10002.09622.822810011.03625.113510022.48633.688210033.94 633.87110045.39635.5999
10063.62644.491410087.75652.557210101.04654.807510122.96659.625910133.92661.2776
10155.83672.120310166.79680.817510177.74688.785410185.61689.095710200.96688.1625
#Mann= 3 , 0 , 0
9799.032    0.12       09799.032    0.12       010200.96    0.12       0
#XS Ineff= 2 , 0
       0                               0
Bank Sta=9799.032,10200.96
Exp/Cntr=0.3,0.1

Type RM Length L Ch R = 1 ,93019.35,246.611300,246.611300,246.611300
XS GIS Cut Line= 6
448520.264016858783144.769944545448564.037288907783176.745888421
448605.937516993783199.847159961448789.063399489783277.150767974
448872.164174416783315.575150444449163.697573871783419.292987176
#Sta/Elev= 30
 9653.29700.5075 9669.29692.02759696.717681.54369731.511669.8173 9755.42663.3498
9787.341651.76239798.325 648.8749809.308647.57469841.838649.78859874.237650.4409
9906.637648.53839917.437646.44219928.237638.66959939.037628.92079948.531622.3441
9960.771615.92859971.797608.23649982.823604.01679993.848603.0444 10026.9603.4416
 10037.9605.673110059.52624.995910080.94626.965310102.35631.667210134.28633.4216
10229.57630.336910303.68631.754510335.44634.457610346.03639.683910355.24640.7113
#Mann= 3 , 0 , 0
 9653.29    0.04       0 9653.29    0.04       010355.24    0.04       0
#XS Ineff= 2 , 0
       0                               0
Bank Sta=9653.29,10355.24
Exp/Cntr=0.3,0.1

Type RM Length L Ch R = 1 ,92772.74,246.611300,246.611300,246.611300
XS GIS Cut Line= 6
448457.399590833783470.521810815448506.899098994783487.505003793
448555.293708985783499.162893136 448969.83115314783570.424171707
449053.302657587783587.886266547449144.246838135 783611.25590843
#Sta/Elev= 30
 9649.04675.51389667.648672.8973 9678.22668.11519699.364661.59859719.991658.8113
9771.195649.69939791.537647.96679801.708646.10349822.004645.27069832.123643.6473
9872.602641.60249902.961 637.5119913.081632.62769923.201626.51159933.321622.6739
 9943.44622.7002 9953.56618.15429973.842 603.5499984.013597.23619994.184592.6031
10014.51  593.8610024.67598.528310044.99613.447310055.15616.652910095.78 615.107
10126.26620.904810166.89622.401210217.95621.739510238.38622.808210350.98623.8334
#Mann= 3 , 0 , 0
 9649.04   0.055       0 9649.04   0.055       010350.98   0.055       0
#XS Ineff= 2 , 0
       0                               0
Bank Sta=9649.04,10350.98
Exp/Cntr=0.3,0.1

Type RM Length L Ch R = 1 ,92526.13,246.611400,246.611400,246.611400
XS GIS Cut Line= 6
448438.351258594783736.490283673448507.706635216  783783.1855904
 448588.99349079783804.251032398448667.991347774 783802.27624546
448913.610408717 783766.57108139449117.555177382783790.659384861
#Sta/Elev= 30
9649.088638.54689662.631633.0937 9683.32627.16919707.311627.43889740.822  632.48
9762.163621.60279782.872623.28959793.002622.08339803.132618.46049817.307611.4029
9843.333605.62959913.642605.65669933.874604.40989954.133598.4904 9984.76582.2259
9994.969578.734510025.61584.770710052.62 584.78510086.19586.761210096.26588.9079
10106.29595.288710126.33597.208810136.35599.894410156.36608.731710166.36609.9692
10226.47610.719210246.58613.078710317.63613.984110327.86616.045210350.94617.3274
#Mann= 3 , 0 , 0
9649.088    0.12       09649.088    0.12       010350.94    0.12       0
#XS Ineff= 2 , 0
       0                               0
Bank Sta=9649.088,10350.94
Exp/Cntr=0.3,0.1

Type RM Length L Ch R = 1 ,92279.52,246.611300,246.611300,246.611300
XS GIS Cut Line= 6
448520.474030733783849.458052502448604.598406859783907.045721102
448766.649291485783975.630503452448888.777251936784041.252100991
449009.517111546784115.359158552449126.865250856784197.757332025
#Sta/Elev= 30
9649.077602.48049773.807601.42629828.313601.92759871.476603.6449 9914.64603.0834
9925.431599.64769936.553591.80799947.741586.78059958.929  585.189970.117582.2731
9981.305577.6394 9988.33576.314110004.18575.293810038.61576.480410050.09574.3936
10061.56575.109110073.13580.148410092.85595.316710096.38596.803710131.26596.9198
10169.63599.843510190.38595.123710206.91593.733410224.69594.470110242.43 592.307
10274.75590.505610286.86591.416610299.23597.369310311.59600.063710350.99601.2325
#Mann= 3 , 0 , 0
9649.077    0.04       09649.077    0.04       010350.99    0.04       0
#XS Ineff= 2 , 0
       0                               0
Bank Sta=9649.077,10350.99
Exp/Cntr=0.3,0.1

Type RM Length L Ch R = 1 ,92032.91,246.611300,246.611300,246.611300
XS GIS Cut Line= 6
448475.882527205783822.520024522448544.909638966783926.120463773
 448611.61630487784108.987445774448644.712678551784167.505545908
448722.667554347 784330.38469132448788.023339818784447.974471993
#Sta/Elev= 30
9649.138 609.5099664.544605.20049689.232601.83389698.802601.42049715.859601.6094
9889.777 599.6149900.269599.02679932.037599.61079942.792594.46229975.463569.8201
9986.893563.60989998.322561.020210016.19560.749310032.95561.185410055.23  560.49
10066.31560.579910082.82562.400410088.48563.346310110.66570.622610121.74573.7084
   10155576.835810166.09579.990210177.17 593.07910188.26596.006310210.43 595.007
10221.68592.370210262.37590.299910290.33 590.90110336.09594.809210350.93595.6055
#Mann= 3 , 0 , 0
9649.138  0.0958       09649.138  0.0958       010350.93  0.0958       0
#XS Ineff= 2 , 0
       0                               0
Bank Sta=9649.138,10350.93
Exp/Cntr=0.3,0.1

Type RM Length L Ch R = 1 , 91786.3,567.349100,567.349100,567.349100
XS GIS Cut Line= 3
448342.032534271783770.305434331448414.949201018784388.360989884
448552.844222188784575.889285624
#Sta/Elev= 30
9639.581633.97159654.377628.37069664.447623.27159674.516616.42349694.655611.9924
9704.724608.22429714.794602.58189734.932599.28669785.279  595.699845.695596.0919
9896.042593.6398 9926.25594.20489966.527564.60119976.597558.91819986.666557.1764
 10006.8556.896210016.87557.504210026.94 561.62810037.01562.393210047.08566.3179
10057.15568.198810127.64567.131610167.91569.390810177.98576.719910198.12588.7655
 10238.4592.177310278.89588.321710419.11585.121110456.35582.936510494.69582.8976
#Mann= 3 , 0 , 0
9639.581   0.049       09639.581   0.049       010494.69   0.049       0
#XS Ineff= 2 , 0
       0                               0
Bank Sta=9639.581,10494.69
Exp/Cntr=0.3,0.1

Type RM Length L Ch R = 1 ,91218.95,326.481800,326.481800,326.481800
XS GIS Cut Line= 2
447717.919453651784035.380026355448405.419453651784955.518915236
#Sta/Elev= 30
9606.001588.31759618.009584.98189642.975581.9333 9734.78578.71939755.323575.8961
9792.772566.39629801.608565.13639835.023565.70649885.144562.27889905.119563.0866
9942.568562.08649980.018553.418710004.98550.318610042.43553.5039 10067.4559.2509
10092.36560.107510117.33564.118610204.71564.625610229.68563.451710292.09563.6638
10366.99566.561910404.44566.312510479.34  568.5610491.82567.912310503.31569.4134
10603.55572.265510679.07578.380110704.03582.9801 10720.5587.406910754.61589.3019
#Mann= 3 , 0 , 0
9606.001    0.12       09606.001    0.12       010754.61    0.12       0
#XS Ineff= 2 , 0
       09881.825        10229.35       0
Bank Sta=9606.001,10754.61
Exp/Cntr=0.3,0.1

Type RM Length L Ch R = 1 ,90892.46,433.377400,433.377400,433.377400
XS GIS Cut Line= 2
447651.947231442784028.435581893447667.572231442784781.907804117
#Sta/Elev= 30
    9605590.28099621.568583.98489651.575576.64249711.588574.82969791.605575.8859
9801.607574.04179811.609568.91479821.611566.59129831.614 565.995 9861.62559.4577
9891.626556.14989941.637554.91029951.639553.49999971.644547.00849981.646545.2069
10001.65544.200410021.65544.904910041.66550.613610071.67553.086410101.67558.3036
10121.68557.980510151.68560.4659 10211.7562.2762 10241.7560.766210271.71555.0863
10281.71 559.60310301.71563.700410321.72 572.60910331.72575.044410358.63576.6838
#Mann= 3 , 0 , 0
    9605  0.0781       0    9605  0.0781       010358.63  0.0781       0
#XS Ineff= 2 , 0
       09867.276        10185.46       0
Bank Sta=9605,10358.63
Exp/Cntr=0.3,0.1

Type RM Length L Ch R = 1 ,90459.09,584.482600,584.482600,584.482600
XS GIS Cut Line= 2
447617.225009203784049.268915251447082.502786994 784488.50502634
#Sta/Elev= 30
9540.361582.77739596.654 573.8319633.829571.57679659.711565.39659672.653560.3162
9706.935551.40159776.182552.89289802.065551.32949815.006552.16369853.829549.1509
9892.653549.29029905.594546.85649927.498545.11299957.359538.22569996.182535.8506
10009.12536.243410022.03546.481510035.01566.488210053.53579.702110073.83596.9943
10085.04601.704710125.59601.982410132.31603.257510151.48 622.21410163.82628.2298
10179.57631.662810195.32637.181710203.24641.044710226.83658.766910232.36659.9982
#Mann= 3 , 0 , 0
9540.361  0.1127       09540.361  0.1127       010232.36  0.1127       0
#XS Ineff= 2 , 0
       09752.156                       0
Bank Sta=9540.361,10232.36
Exp/Cntr=0.3,0.1

Type RM Length L Ch R = 1 , 89874.6,706.174800,706.174800,706.174800
XS GIS Cut Line= 6
447565.986901343 783920.80462262447410.348080039783840.095152304
447255.309708387783784.340042979447229.681130409783796.323282033
447174.516675949783853.088359684446790.402092546784041.890443027
#Sta/Elev= 30
9604.327639.00229636.436642.33269719.412643.31489774.637641.23689806.943 624.167
9817.661622.00549860.532 591.341 9871.25587.53629881.967578.36849903.403563.4389
9914.121559.24919935.017546.55329944.857542.6584 9971.16526.45049994.826524.8653
10025.13525.5523 10039.8532.346610052.56536.026810074.93538.503310141.78538.4323
10230.92542.835310242.07545.448710284.21565.569110306.88573.149410331.21575.1604
10353.49574.705610375.78590.483710431.49615.796210464.92620.331410481.19617.8475
#Mann= 3 , 0 , 0
9604.327  0.0969       09604.327  0.0969       010481.19  0.0969       0
#XS Ineff= 2 , 0
       0                               0
Bank Sta=9604.327,10481.19
Exp/Cntr=0.3,0.1

Type RM Length L Ch R = 1 ,89168.43,798.318700,798.318700,798.318700
XS GIS Cut Line= 6
447462.204754651783837.174007833447208.298504591783749.283382818
447141.024199039783703.710466176447048.793296248783607.139285624
446992.822009414783566.254263222446550.384731442783155.605720818
#Sta/Elev= 30
9153.808647.92499193.179647.23799221.595 639.5099246.089628.37869277.836 600.003
    9299 590.3279330.747568.35479351.911559.5538 9405.02555.01699422.496546.3182
9462.715537.06569474.794 536.8439501.454 546.2199529.626546.48999584.869555.6381
9626.422557.22149703.908552.0871    9765554.75999835.775533.83249926.335530.9999
9966.816522.40289983.604515.1618 10007.3513.805710043.18518.652110088.26565.8893
10117.65578.838110128.74580.101410207.02552.0378 10251.7 544.02910310.38524.7589
#Mann= 3 , 0 , 0
9153.808  0.0883       09153.808  0.0883       010310.38  0.0883       0
#XS Ineff= 2 , 0
       0                               0
Bank Sta=9153.808,10310.38
Exp/Cntr=0.3,0.1

Type RM Length L Ch R = 1 ,88370.11,488.026300,488.026300,488.026300
XS GIS Cut Line= 6
447542.085049093783823.740409613447427.498294324 783724.86458376
447377.389086068 783657.32530202 447352.49867481783606.417646885
  447330.7173886783480.240675211447336.843064785783303.175165236
#Sta/Elev= 30
9749.068 621.0159758.132623.07469770.925627.7618 9795.15631.90069811.184  628.94
9833.239619.90419842.574614.60689857.521602.5598 9875.61590.50729889.882579.6141
9913.233570.2328 9926.05561.42979938.867 548.5619951.685538.03989955.193530.9153
9963.815509.94159970.673505.26159975.686 502.4539984.796500.372310010.21499.2078
10021.23500.653710043.01506.698210074.43518.935810125.34528.290610145.38535.1351
10165.42545.848910195.44557.2917 10285.5579.025110305.51 588.24210347.37600.6839
#Mann= 3 , 0 , 0
9749.068    0.12       09749.068    0.12       010347.37    0.12       0
#XS Ineff= 2 , 0
       0                               0
Bank Sta=9749.068,10347.37
Exp/Cntr=0.3,0.1

Type RM Length L Ch R = 1 ,87882.09,488.026400,488.026400,488.026400
XS GIS Cut Line= 6
447994.794194957783573.761391918447945.491290225783546.426666803
447895.376491365 783513.96605768 447772.71365711783419.590042677
447739.216370869783387.571671349447614.951980851783250.944422495
#Sta/Elev= 30
9749.028583.71899771.661578.97929805.987 574.0469817.901568.31159829.816560.9016
9844.814550.32239863.209535.47829877.969524.69529890.361518.49469902.753513.6597
9915.145509.87279940.454507.27059953.172503.9177 9965.89 497.9779991.326494.1857
    9999493.825710016.96495.199810030.58495.298310041.02 497.18510058.24503.2408
10072.61506.158510083.03510.5874 10087.7511.637210102.79513.314210148.08516.1621
10176.48  520.0310187.19522.118310193.09523.640110221.99533.878910250.96547.2477
#Mann= 3 , 0 , 0
9749.028    0.12       09749.028    0.12       010250.96    0.12       0
#XS Ineff= 2 , 0
       0                               0
Bank Sta=9749.028,10250.96
Exp/Cntr=0.3,0.1

Type RM Length L Ch R = 1 ,87394.06,488.026300,488.026300,488.026300
XS GIS Cut Line= 6
448009.141862168782885.168973344 447953.39490068782911.675764183
447905.495229198782931.541795409447743.711041445782989.594399934
447664.618636242783011.664746657447533.257935066 783039.92089212
#Sta/Elev= 30
9749.019545.61099764.678543.33469786.823538.18069819.424532.19259841.487529.7644
9852.313526.56299873.768512.94419895.046504.01419905.685 501.7699916.324501.2795
9926.963 498.9519937.602494.0592 9958.88490.02389969.519490.01419990.797484.7239
   10012484.270110022.56484.677710033.13488.290210043.54 494.81310053.92503.1373
 10064.3513.875310085.06527.831910105.83544.375610116.21551.579210126.44557.4199
 10146.9565.383610177.59573.905510198.05588.5733 10218.5599.265510250.97619.2884
#Mann= 3 , 0 , 0
9749.019    0.12       09749.019    0.12       010250.97    0.12       0
#XS Ineff= 2 , 0
       0                               0
Bank Sta=9749.019,10250.97
Exp/Cntr=0.3,0.1

Type RM Length L Ch R = 1 ,86906.03,488.026400,488.026400,488.026400
XS GIS Cut Line= 6
447481.577437452782465.033281294447477.808367938782634.982705751
447505.272140349782785.941177911447510.144605683782841.071744241
447504.262267921782899.692473722447483.957402871782960.035122499
#Sta/Elev= 30
9749.051552.33489769.057 542.7279789.096528.54459809.135516.29369829.174512.9308
9839.188512.85879849.188 514.8189869.188513.70139879.189507.51019889.199 498.558
9919.232481.6678 9929.31479.87229959.543479.37239969.621479.58179990.037481.8247
10010.49480.313710020.71483.907410030.93490.463310071.81521.398610081.87525.5447
10101.95531.855910132.05538.776710152.07546.165610162.15548.933310172.26552.8697
10182.38558.709210203.07567.242610213.48572.888310234.62581.824910250.88587.0572
#Mann= 3 , 0 , 0
9749.051    0.12       09749.051    0.12       010250.88    0.12       0
#XS Ineff= 2 , 0
       0                               0
Bank Sta=9749.051,10250.88
Exp/Cntr=0.3,0.1

Type RM Length L Ch R = 1 ,86418.01,488.026300,488.026300,488.026300
XS GIS Cut Line= 6
446954.629056271782432.552525744446966.825046182782642.564045034
447005.279860299782782.401410067447129.049699808783020.286702966
447165.490019725783047.909687374447244.336207282783064.919497975
#Sta/Elev= 30
9624.056510.35499656.512 504.347 9686.52494.34149696.523493.04069786.687487.5834
9816.897484.27749837.069484.77419877.701 480.6819898.248482.51019929.415 481.858
9950.433477.93489961.257477.03439972.082473.79049994.082 471.52310005.23471.6812
10016.42473.7371 10038.8494.592310061.17504.703310105.38531.428410116.43536.7424
10138.54544.120710160.65555.852410194.17563.937710205.83 565.12610217.48564.4233
10256.96570.854210270.63573.688210304.96584.654910346.42591.892910375.97599.8021
#Mann= 3 , 0 , 0
9624.056  0.0805       09624.056  0.0805       010375.97  0.0805       0
#XS Ineff= 2 , 0
       0                               0
Bank Sta=9624.056,10375.97
Exp/Cntr=0.3,0.1

Type RM Length L Ch R = 1 ,85929.98,488.026400,488.026400,488.026400
XS GIS Cut Line= 6
446668.992632329782406.086488456446634.451951534782588.278387055
446614.131994575782662.258314222446573.092327446782769.378772482
 446489.18370381782935.573156387446419.670032352783196.331993952
#Sta/Elev= 30
9624.049 493.1899643.231491.92279704.083490.73849714.225489.46039755.083487.0603
  9765.3 485.9189795.954484.41029899.778480.99139921.026477.43859931.649478.3183
9942.273478.02249963.635472.99639985.367465.563510007.21465.483710029.32467.1385
10040.37471.295910054.94481.438810062.63485.804210066.03486.174210141.49486.2932
10228.01487.361710248.71488.826910279.75489.487310321.15492.6153 10352.2498.5603
 10393.6513.451610414.29524.110410424.64530.645610434.99532.665110457.07533.0621
#Mann= 3 , 0 , 0
9624.049   0.083       09624.049   0.083       010457.07   0.083       0
#XS Ineff= 2 , 0
       0                10096.01       0
Bank Sta=9624.049,10457.07
Exp/Cntr=0.3,0.1

Type RM Length L Ch R = 1 ,85441.95,488.026300,488.026300,488.026300
XS GIS Cut Line= 6
446069.867002904782267.926071644446072.189927965782439.397286177
446116.697976738782657.092027724446218.755850226782862.958449036
446243.176558286782936.275717244446234.774199039783316.123660624
#Sta/Elev= 30
9624.044579.32419631.137 577.2959661.216579.5267 9701.25558.24439711.258547.7804
9721.266544.69019741.284544.4948 9771.38526.93289832.002514.29869872.563509.9579
9903.218493.15689944.207480.05899974.948461.06939995.442458.539610016.03459.9378
10026.43 465.52910047.27469.353410184.14477.165310261.58476.534210304.01478.8104
10374.84476.900910484.86480.619310524.87479.553910544.88474.502710554.88475.1582
10584.89481.854610604.89489.351310674.91523.686710694.91529.131410706.04529.1304
#Mann= 3 , 0 , 0
9624.044    0.12       09624.044    0.12       010706.04    0.12       0
#XS Ineff= 2 , 0
       0                10318.48       0
Bank Sta=9624.044,10706.04
Exp/Cntr=0.3,0.1

Type RM Length L Ch R = 1 ,84953.93,488.026300,488.026300,488.026300
XS GIS Cut Line= 6
445849.860493854782731.491167157445882.164504948 782849.89622986
445889.114607341782931.850878263 445881.38357768  782951.9921545
445827.688732541783029.665429477445768.360424392783199.310151329
#Sta/Elev= 30
 9749.15524.72259766.771511.15329784.182500.46579801.056488.94819815.502481.6986
9836.064 473.3989846.345471.51299866.907470.23319887.215465.38389897.327465.2297
 9907.44463.99169927.592459.45439937.605455.38949968.365457.34449980.116453.1991
 9993.18452.0413 10006.4 454.18610019.43458.807810024.56462.240510034.46470.8154
10054.73483.290710065.91491.638610076.86498.5896 10087.6507.404510109.09523.3805
10141.24549.793210151.76556.583310172.79574.1469 10183.3582.054610250.92619.7339
#Mann= 3 , 0 , 0
 9749.15    0.12       0 9749.15    0.12       010250.92    0.12       0
#XS Ineff= 2 , 0
       0                               0
Bank Sta=9749.15,10250.92
Exp/Cntr=0.3,0.1

Type RM Length L Ch R = 1 , 84465.9,572.692600,572.692600,572.692600
XS GIS Cut Line= 6
445478.659527964782529.117724038445460.127742036782623.248963687
 445451.08858149782759.643647682445438.386467067782870.161698248
445424.160791088782945.421409329445403.550313585 783024.07553576
#Sta/Elev= 30
9749.058620.86149765.442615.40819786.075602.43819794.192596.00349816.564576.4737
9836.781557.85629856.896 541.274 9876.94527.44729886.962518.39299896.984511.1692
9907.006502.82619937.072473.83999947.094463.66159957.116457.57089967.138454.6058
 9977.16449.25129987.198446.533610007.32446.873310017.38450.010210027.45458.2847
10037.52471.066410047.59482.538110057.66492.797310067.73504.451610077.79512.9532
10097.98532.165310148.87574.329810169.65586.427410189.89599.283410250.96630.4372
#Mann= 3 , 0 , 0
9749.058    0.12       09749.058    0.12       010250.96    0.12       0
#XS Ineff= 2 , 0
       0                               0
Bank Sta=9749.058,10250.96
Exp/Cntr=0.3,0.1

Type RM Length L Ch R = 1 ,83893.21,403.360100,403.360100,403.360100
XS GIS Cut Line= 2
444995.868964285782550.809247002444718.715171248782889.908382818
#Sta/Elev= 30
 9825.59508.80479831.003507.66539858.567497.52719882.663485.21289895.579480.9593
9905.972 476.3639908.494474.82199921.409462.92839934.324454.34679947.239450.3565
9960.154444.9375 9973.07442.72889985.985442.607810011.82443.343310024.73 444.703
10037.65454.669110050.56466.520710063.48 476.28810076.39481.214510095.59493.3424
10102.22496.676910115.14499.659910128.05508.359810140.97512.8335 10158.8 514.731
10179.71527.393310192.63 532.93210231.37555.392910253.61566.418610263.54570.4588
#Mann= 3 , 0 , 0
 9825.59    0.12       0 9825.59    0.12       010263.54    0.12       0
#XS Ineff= 2 , 0
       0                               0
Bank Sta=9825.59,10263.54
Exp/Cntr=0.3,0.1

Type RM Length L Ch R = 1 ,83489.85,488.026300,488.026300,488.026300
XS GIS Cut Line= 6
444995.204846733782518.761810979 444931.82578949782516.066596442
444880.024381128 782488.58882573444746.815149331782311.767454183
444684.610811747782262.843029284444616.115913513782227.512954566
#Sta/Elev= 30
9749.076509.99649779.341505.93389789.351503.91119799.446500.1147  9816.1490.5615
9841.887472.92729853.722464.00789865.835457.80839878.742 455.0279892.435454.9306
9906.076451.95469943.838448.37869957.131443.81199978.914439.07259990.361435.4657
10013.59 434.95610017.25435.842610037.36446.362310049.99455.409810067.91475.2751
10090.09496.468510104.81512.577610120.01527.344410136.51541.884610170.03 568.877
10184.88578.471710196.45589.521210209.48600.374910230.08615.882510250.91633.1326
#Mann= 3 , 0 , 0
9749.076    0.12       09749.076    0.12       010250.91    0.12       0
#XS Ineff= 2 , 0
       0                               0
Bank Sta=9749.076,10250.91
Exp/Cntr=0.3,0.1

Type RM Length L Ch R = 1 ,83001.82,472.726200,472.726200,472.726200
XS GIS Cut Line= 6
445458.191011387782319.284987541445400.459886416782300.604791187
445329.855133057782258.388212964445240.519695529782182.247274482
445178.060318794782139.397292859445056.596060197  782027.2770787
#Sta/Elev= 30
9749.114 619.4339762.667622.35659767.779 621.6169773.046619.9367 9797.29607.3596
9809.898596.10349827.305582.54639843.676566.62889862.212545.41479874.164528.5648
9886.116509.51029892.265501.82719913.806478.26579929.896457.46129936.757449.6485
9962.287430.47499975.441426.4257    9999425.960910028.19 430.14710041.95434.0939
10064.29437.851210076.39440.9804 10092.1447.4249   10117453.457410130.61460.2585
10171.43473.297710198.65478.416810225.87488.959810239.48 495.81910250.92502.8634
#Mann= 3 , 0 , 0
9749.114    0.12       09749.114    0.12       010250.92    0.12       0
#XS Ineff= 2 , 0
       0                               0
Bank Sta=9749.114,10250.92
Exp/Cntr=0.3,0.1

Type RM Length L Ch R = 1 , 82529.1,503.326500,503.326500,503.326500
XS GIS Cut Line= 6
445631.745155931781727.290386826445578.185508102781746.573213577
445483.526844114781768.319241747445388.235291302781778.385322228
445355.813640952781778.873679474445120.190865695781861.262549505
#Sta/Elev= 30
 9747.89608.84769786.944570.15549839.211521.56479859.764  502.779880.135486.5547
9900.506468.15769910.594458.24979920.665449.78029940.806438.05429960.945434.0021
9970.981431.01989991.053423.312710011.09422.948110021.09 422.99410031.14424.6721
10041.73427.851510062.92440.860310073.51448.287510084.11454.2544 10094.7456.6067
10126.48465.955510137.08467.084410158.26473.337910190.04480.523310200.64484.0454
10211.23486.286710221.83 489.77710243.01500.594410260.91508.368110279.89514.3919
#Mann= 3 , 0 , 0
 9747.89    0.12       0 9747.89    0.12       010279.89    0.12       0
#XS Ineff= 2 , 0
       0                               0
Bank Sta=9747.89,10279.89
Exp/Cntr=0.3,0.1

Type RM Length L Ch R = 1 ,82025.77,488.026400,488.026400,488.026400
XS GIS Cut Line= 6
445061.531690383781273.326732009445039.021107471781404.661660264
445029.428201138781588.310217737445021.836917285781649.720465019
445004.450204135781706.013891991444970.380394515781759.660317817
#Sta/Elev= 30
9749.028464.63219760.926466.9859 9771.12472.32419781.313480.05119791.506491.7542
9801.699501.59999811.893507.51019822.086507.36369832.191497.74329842.287486.3833
9852.383475.8064 9882.67438.30879892.701428.54779912.764419.18229922.795416.6389
9932.826 417.1679952.871416.2401 10002.9415.420410012.91415.892710022.92419.2363
10042.94429.221810052.94 432.12310083.02434.365210133.61434.6148 10154.2435.5729
10175.46438.3062 10186.1438.723510197.45440.136410220.32449.438910250.91468.9107
#Mann= 3 , 0 , 0
9749.028    0.12       09749.028    0.12       010250.91    0.12       0
#XS Ineff= 2 , 0
       0                               0
Bank Sta=9749.028,10250.91
Exp/Cntr=0.3,0.1

Type RM Length L Ch R = 1 ,81537.74,488.026300,488.026300,488.026300
XS GIS Cut Line= 6
444611.398831567781181.463461772444585.874204994781291.625455772
444561.581384633781426.350761269444537.333460907781553.232870319
444522.210623874781610.278410397 444500.57410966781670.251231128
#Sta/Elev= 30
9749.022626.45749773.182606.92759783.447599.49389803.976581.06949814.241574.2703
9821.673568.22849855.301537.91379865.531525.93049875.692519.10989885.854509.8652
9896.015494.15119906.176477.25879926.499446.6462 9936.66436.42169946.821424.2387
9967.144  409.439977.305407.799310017.99407.989310038.35412.629710058.71413.5175
10087.32426.751610099.43430.777710109.62435.9657 10119.8439.492910130.01444.2617
10161.04461.676410171.39465.678110187.19470.447910202.84473.157210250.95484.9841
#Mann= 3 , 0 , 0
9749.022    0.12       09749.022    0.12       010250.95    0.12       0
#XS Ineff= 2 , 0
       0                               0
Bank Sta=9749.022,10250.95
Exp/Cntr=0.3,0.1

Type RM Length L Ch R = 1 ,81049.72,488.026300,488.026300,488.026300
XS GIS Cut Line= 6
444286.591693658781026.142171688444249.125916773 781088.47716681
444213.645456794781141.276056352444129.931420737781257.600995656
444043.466098945781369.742168316443996.611581934781435.450677946
#Sta/Elev= 30
 9749.02 532.0939794.357502.22329817.691492.26559841.655478.22329865.751461.2323
9877.799448.81019914.638 419.8549926.979412.75599951.309406.54769964.002 402.292
9968.374401.677510000.99401.350810019.91401.532410038.02405.876810063.28409.8868
 10075.9413.260310088.53413.248910101.16411.778410126.41415.154310135.02414.9825
10151.39420.5589 10164.3426.700410176.74431.684710184.87433.2619 10201.3432.0696
10213.59426.738210219.31426.428510225.87426.924410238.15423.238210250.99426.7651
#Mann= 3 , 0 , 0
 9749.02    0.12       0 9749.02    0.12       010250.99    0.12       0
#XS Ineff= 2 , 0
       0                               0
Bank Sta=9749.02,10250.99
Exp/Cntr=0.3,0.1

Type RM Length L Ch R = 1 ,80561.69,488.026400,488.026400,488.026400
XS GIS Cut Line= 6
443731.349822261780754.040870074443726.207720331780846.817423178
443728.125178027780921.621894897443753.795676044781075.337600057
443758.456861239781130.509029114443751.040998449781252.964774884
#Sta/Elev= 30
9749.065521.85699760.041523.80429770.056522.62499780.071520.27899800.102512.8984
9841.984488.14819870.176 469.8339880.179458.78689890.182 456.9139920.215434.9889
9950.432410.79789960.505404.19699990.935392.915410001.07392.628810011.26392.6672
10031.65395.656710052.04395.079210062.23 400.04510072.43401.3272 10092.5406.5339
10102.54407.092810122.61410.150310132.63414.545710152.63434.105910182.64458.5371
10192.67 470.25910202.72476.531510232.86 499.58310242.91505.328410250.92 508.576
#Mann= 3 , 0 , 0
9749.065    0.12       09749.065    0.12       010250.92    0.12       0
#XS Ineff= 2 , 0
       0                               0
Bank Sta=9749.065,10250.92
Exp/Cntr=0.3,0.1
